--- U102-00-00.prj (project) ---

Proj Title=U102-00-00 (Update)
Current Plan=p01
Default Exp/Contr=0.3,0.1
English Units
Geom File=g01
Flow File=f01
Flow File=f02
Plan File=p01
Plan File=p02
Y Axis Title=Elevation
X Axis Title(PF)=Main Channel Distance
X Axis Title(XS)=Station
BEGIN DESCRIPTION:
Bear Creek (U102-00-00)
(Flood Hazard & Floodway) Model
10-, 2-, 1-, and 0.2% Events
FILENAME: U102_00_00.prj
PREPARED BY:  LAN                                 DATE: 03/13/2014
REVIEWED BY: LJA                                   DATE: 03/14/2014
STATUS: Final
ADDICKS WATERSHED MODEL UPDATE
HARRIS COUNTY, TEXAS
Update1:
The effective FEMA hydraulic model for unit number U102-00-00 has been updated by FEMA LOMR 20-06-2070P with an effective date of XX/XX/XXXX.
Update2:
The effective FEMA hydraulic model for unit number U102-00-00 has been updated by FEMA LOMR 20-06-2933P with an effective date of 05/17/2021.
END DESCRIPTION:
DSS File=dss
DSS Export Rating Curves= 0
DSS Export Rating Curve Sorted= 0
DSS Export Volume Flow Curves= 0
DXF OffsetX= 0
DXF OffsetY= 0
DXF ScaleX= 1
DXF ScaleY= 10

--- U102-00-00.p01 (plan) ---

Plan Title=Effective Multi-Profile 2021
Program Version=4.10
Short Identifier=Eff+LOMR MP
Geom File=g01
Flow File=f01
Subcritical Flow
K Sum by GR= 0
Std Step Tol= 0.01
Critical Tol= 0.01
Num of Std Step Trials= 20
Max Error Tol= 0.3
Flow Tol Ratio= 0.001
Split Flow NTrial= 30
Split Flow Tol= 0.02
Split Flow Ratio= 0.02
Log Output Level= 0
Friction Slope Method= 1
Unsteady Friction Slope Method= 2
Unsteady Bridges Friction Slope Method= 1
Parabolic Critical Depth
Global Vel Dist= 0 , 0 , 0
Global Log Level= 0
CheckData=True
Encroach Param=-1 ,0,0, 0
BEGIN DESCRIPTION:
FEMA Effective Multi-Profile November 2019 + LOMR 20-06-2070P
END DESCRIPTION:
Computation Interval=1HOUR
Output Interval=1HOUR
Run HTab= 0
Run UNet= 0
Run PostProcess= 0
Run WQNet= 0
UNET Theta= 1
UNET Theta Warmup= 1
UNET ZTol= 0.02
UNET ZSATol= 0.05
UNET MxIter= 20
UNET MaxInSteps= 0
UNET DtIC= 0
UNET DtMin= 0
UNET MaxCRTS= 20
UNET WFStab= 2
UNET SFStab= 1
UNET WFX= 1
UNET SFX= 1
UNET DSS MLevel= 4
UNET DZMax Abort= 100
UNET Convert EG Bridges= 0
UNET Use Existing IB Tables=-1
UNET Froude Reduction=False
UNET Froude Limit= 1
UNET Froude Power= 10
UNET Time Slicing=0,0, 5
UNET Junction Losses=0
Instantaneous Interval=1HOUR
Write IC File= 0
Write IC File at Sim End=0
Echo Input=False
Echo Parameters=False
Echo Output=False
Write Detailed= 0
WQ AD Non Conservative
WQ ULTIMATE=-1
WQ Max Comp Step=1HOUR
WQ Output Interval=15MIN
WQ Output Selected Increments= 0
WQ Output face flow=0
WQ Output face velocity=0
WQ Output face area=0
WQ Output face dispersion=0
WQ Output cell volume=0
WQ Output cell surface area=0
WQ Output cell continuity=0
WQ Output cumulative cell continuity=0
WQ Output face conc=0
WQ Output face dconc_dx=0
WQ Output face courant=0
WQ Output face peclet=0
WQ Output face adv mass=0
WQ Output face disp mass=0
WQ Output cell mass=0
WQ Output cell source sink temp=0
WQ Output cell source sink nsm=0
WQ Output MaxMinRange=-1
WQ Daily Max Min Mean=-1
WQ Daily Range=0
WQ Daily Time=0
WQ Create Restart=0
WQ Fixed Restart=0
WQ System Summary=0
WQ Use Fixed Temperature=0
Sorting and Armoring Iterations= 10
XS Update Threshold= 0.02
Hydraulics Update Threshold= 0.02
Energy Slope Method= 1
Volume Change Method= 0
XS Weighting Method= 0
Number of US Weighted Cross Sections= 1
Number of DS Weighted Cross Sections= 1
Upstream XS Weight=0.25
Main XS Weight=0.5
Downstream XS Weight=0.25
Number of DS XS's Weighted with US Boundary= 1
Upstream Boundary Weight= 1
Weight of XSs Associated with US Boundary= 0
Number of US XS's Weighted with DS Boundary= 1
Downstream Boundary Weight= 0.5
Weight of XSs Associated with DS Boundary= 0.5
Sediment Output Level= 4
Mass or Volume Output= 0
Output Increment Type= 1
Profile and TS Output Increment= 10
XS Output Flag= 0
XS Output Increment= 10
Disregard all LS=0
Disregard all Conn=0
Disregard all Breaches=0
Disregard all Pumps=0

--- U102-00-00.p02 (plan) ---

Plan Title=Effective FW 2021
Program Version=4.10
Short Identifier=PostPrj+LOMR FW
Geom File=g01
Flow File=f02
Subcritical Flow
K Sum by GR= 0
Std Step Tol= 0.01
Critical Tol= 0.01
Num of Std Step Trials= 20
Max Error Tol= 0.3
Flow Tol Ratio= 0.001
Split Flow NTrial= 30
Split Flow Tol= 0.02
Split Flow Ratio= 0.02
Log Output Level= 0
Friction Slope Method= 1
Unsteady Friction Slope Method= 2
Unsteady Bridges Friction Slope Method= 1
Parabolic Critical Depth
Global Vel Dist= 10 , 1 , 10
Vel Dist Location=U102-00-00      ,U102-00-00_0197 ,82591.49, 10 , 1 , 10
Vel Dist Location=U102-00-00      ,U102-00-00_0197 ,81731.22, 10 , 1 , 10
Vel Dist Location=U102-00-00      ,U102-00-00_0197 ,81073.43, 10 , 1 , 10
Vel Dist Location=U102-00-00      ,U102-00-00_0197 ,80119.4 , 10 , 1 , 10
Vel Dist Location=U102-00-00      ,U102-00-00_0197 ,78904.98, 10 , 1 , 10
Vel Dist Location=U102-00-00      ,U102-00-00_0197 ,78687.62, 10 , 1 , 10
Vel Dist Location=U102-00-00      ,U102-00-00_0197 ,78672.98, 10 , 1 , 10
Vel Dist Location=U102-00-00      ,U102-00-00_0197 ,78654.82, 10 , 1 , 10
Vel Dist Location=U102-00-00      ,U102-00-00_0197 ,78422.85, 10 , 1 , 10
Vel Dist Location=U102-00-00      ,U102-00-00_0197 ,77603.52, 10 , 1 , 10
Vel Dist Location=U102-00-00      ,U102-00-00_0197 ,76413.3 , 10 , 1 , 10
Vel Dist Location=U102-00-00      ,U102-00-00_0197 ,74758.11, 10 , 1 , 10
Vel Dist Location=U102-00-00      ,U102-00-00_0197 ,74313.45, 10 , 1 , 10
Vel Dist Location=U102-00-00      ,U102-00-00_0197 ,73108.58, 10 , 1 , 10
Vel Dist Location=U102-00-00      ,U102-00-00_0197 ,71949.68, 10 , 1 , 10
Vel Dist Location=U102-00-00      ,U102-00-00_0197 ,71324.16, 10 , 1 , 10
Vel Dist Location=U102-00-00      ,U102-00-00_0197 ,69870.13, 10 , 1 , 10
Vel Dist Location=U102-00-00      ,U102-00-00_0197 ,69031.07, 10 , 1 , 10
Vel Dist Location=U102-00-00      ,U102-00-00_0197 ,68924.32, 10 , 1 , 10
Vel Dist Location=U102-00-00      ,U102-00-00_0197 ,68899.68, 10 , 1 , 10
Vel Dist Location=U102-00-00      ,U102-00-00_0197 ,68877.77, 10 , 1 , 10
Vel Dist Location=U102-00-00      ,U102-00-00_0197 ,68441.07, 10 , 1 , 10
Vel Dist Location=U102-00-00      ,U102-00-00_0197 ,67625.08, 10 , 1 , 10
Vel Dist Location=U102-00-00      ,U102-00-00_0197 ,66253.16, 10 , 1 , 10
Vel Dist Location=U102-00-00      ,U102-00-00_0197 ,65864.54, 10 , 1 , 10
Vel Dist Location=U102-00-00      ,U102-00-00_0197 ,65139.42, 10 , 1 , 10
Vel Dist Location=U102-00-00      ,U102-00-00_0197 ,64170.07, 10 , 1 , 10
Vel Dist Location=U102-00-00      ,U102-00-00_0197 ,63598.3 , 10 , 1 , 10
Vel Dist Location=U102-00-00      ,U102-00-00_0197 ,63543.31, 10 , 1 , 10
Vel Dist Location=U102-00-00      ,U102-00-00_0197 ,63482.86, 10 , 1 , 10
Vel Dist Location=U102-00-00      ,U102-00-00_0197 ,63435.61, 10 , 1 , 10
Vel Dist Location=U102-00-00      ,U102-00-00_0197 ,63182.11, 10 , 1 , 10
Vel Dist Location=U102-00-00      ,U102-00-00_0197 ,62613.3 , 10 , 1 , 10
Vel Dist Location=U102-00-00      ,U102-00-00_0197 ,61507.56, 10 , 1 , 10
Vel Dist Location=U102-00-00      ,U102-00-00_0197 ,60176.11, 10 , 1 , 10
Vel Dist Location=U102-00-00      ,U102-00-00_0197 ,59168.92, 10 , 1 , 10
Vel Dist Location=U102-00-00      ,U102-00-00_0197 ,58086.16, 10 , 1 , 10
Vel Dist Location=U102-00-00      ,U102-00-00_0197 ,57213.66, 10 , 1 , 10
Vel Dist Location=U102-00-00      ,U102-00-00_0197 ,57093.08, 10 , 1 , 10
Vel Dist Location=U102-00-00      ,U102-00-00_0197 ,57037.9 , 10 , 1 , 10
Vel Dist Location=U102-00-00      ,U102-00-00_0197 ,56832.31, 10 , 1 , 10
Vel Dist Location=U102-00-00      ,U102-00-00_0197 ,56666.18, 10 , 1 , 10
Vel Dist Location=U102-00-00      ,U102-00-00_0197 ,56470.21, 10 , 1 , 10
Vel Dist Location=U102-00-00      ,U102-00-00_0197 ,56194.89, 10 , 1 , 10
Vel Dist Location=U102-00-00      ,U102-00-00_0197 ,56132.66, 10 , 1 , 10
Vel Dist Location=U102-00-00      ,U102-00-00_0197 ,55887.13, 10 , 1 , 10
Vel Dist Location=U102-00-00      ,U102-00-00_0197 ,55580.36, 10 , 1 , 10
Vel Dist Location=U102-00-00      ,U102-00-00_0197 ,55351.98, 10 , 1 , 10
Vel Dist Location=U102-00-00      ,U102-00-00_0197 ,54885.61, 10 , 1 , 10
Vel Dist Location=U102-00-00      ,U102-00-00_0197 ,54244.41, 10 , 1 , 10
Vel Dist Location=U102-00-00      ,U102-00-00_0197 ,53109.38, 10 , 1 , 10
Vel Dist Location=U102-00-00      ,U102-00-00_0197 ,52414.93, 10 , 1 , 10
Vel Dist Location=U102-00-00      ,U102-00-00_0197 ,52204.51, 10 , 1 , 10
Vel Dist Location=U102-00-00      ,U102-00-00_0197 ,52104.96, 10 , 1 , 10
Vel Dist Location=U102-00-00      ,U102-00-00_0197 ,52072.36, 10 , 1 , 10
Vel Dist Location=U102-00-00      ,U102-00-00_0197 ,52014.66, 10 , 1 , 10
Vel Dist Location=U102-00-00      ,U102-00-00_0197 ,51929.68, 10 , 1 , 10
Vel Dist Location=U102-00-00      ,U102-00-00_0197 ,51782.55, 10 , 1 , 10
Vel Dist Location=U102-00-00      ,U102-00-00_0197 ,51146.17, 10 , 1 , 10
Vel Dist Location=U102-00-00      ,U102-00-00_0197 ,51047.25, 10 , 1 , 10
Vel Dist Location=U102-00-00      ,U102-00-00_0197 ,50998.88, 10 , 1 , 10
Vel Dist Location=U102-00-00      ,U102-00-00_0197 ,49965.56, 10 , 1 , 10
Vel Dist Location=U102-00-00      ,U102-00-00_0197 ,48859.02, 10 , 1 , 10
Vel Dist Location=U102-00-00      ,U102-00-00_0197 ,47847.21, 10 , 1 , 10
Vel Dist Location=U102-00-00      ,U102-00-00_0197 ,47111.71, 10 , 1 , 10
Vel Dist Location=U102-00-00      ,U102-00-00_0197 ,46984.47, 10 , 1 , 10
Vel Dist Location=U102-00-00      ,U102-00-00_0197 ,46926.72, 10 , 1 , 10
Vel Dist Location=U102-00-00      ,U102-00-00_0197 ,46873.4 , 10 , 1 , 10
Vel Dist Location=U102-00-00      ,U102-00-00_0197 ,46507.83, 10 , 1 , 10
Vel Dist Location=U102-00-00      ,U102-00-00_0197 ,46401.06, 10 , 1 , 10
Vel Dist Location=U102-00-00      ,U102-00-00_0197 ,46387.11, 10 , 1 , 10
Vel Dist Location=U102-00-00      ,U102-00-00_0197 ,46369.31, 10 , 1 , 10
Vel Dist Location=U102-00-00      ,U102-00-00_0197 ,46304.02, 10 , 1 , 10
Vel Dist Location=U102-00-00      ,U102-00-00_0197 ,45910.1 , 10 , 1 , 10
Vel Dist Location=U102-00-00      ,U102-00-00_0197 ,45379.92, 10 , 1 , 10
Vel Dist Location=U102-00-00      ,U102-00-00_0197 ,44394.45, 10 , 1 , 10
Vel Dist Location=U102-00-00      ,U102-00-00_0197 ,43344.77, 10 , 1 , 10
Vel Dist Location=U102-00-00      ,U102-00-00_0197 ,42393.07, 10 , 1 , 10
Vel Dist Location=U102-00-00      ,U102-00-00_0197 ,41585.04, 10 , 1 , 10
Vel Dist Location=U102-00-00      ,U102-00-00_0197 ,41483.83, 10 , 1 , 10
Vel Dist Location=U102-00-00      ,U102-00-00_0197 ,41408.37, 10 , 1 , 10
Vel Dist Location=U102-00-00      ,U102-00-00_0197 ,41354.38, 10 , 1 , 10
Vel Dist Location=U102-00-00      ,U102-00-00_0197 ,40963.29, 10 , 1 , 10
Vel Dist Location=U102-00-00      ,U102-00-00_0197 ,40319   , 10 , 1 , 10
Vel Dist Location=U102-00-00      ,U102-00-00_0197 ,39300.46, 10 , 1 , 10
Vel Dist Location=U102-00-00      ,U102-00-00_0197 ,38178.64, 10 , 1 , 10
Vel Dist Location=U102-00-00      ,U102-00-00_0197 ,37416.59, 10 , 1 , 10
Vel Dist Location=U102-00-00      ,U102-00-00_0197 ,37245.13, 10 , 1 , 10
Vel Dist Location=U102-00-00      ,U102-00-00_0197 ,37207.97, 10 , 1 , 10
Vel Dist Location=U102-00-00      ,U102-00-00_0197 ,37157.18, 10 , 1 , 10
Vel Dist Location=U102-00-00      ,U102-00-00_0197 ,36534.81, 10 , 1 , 10
Vel Dist Location=U102-00-00      ,U102-00-00_0197 ,35899.56, 10 , 1 , 10
Vel Dist Location=U102-00-00      ,U102-00-00_0197 ,34772.93, 10 , 1 , 10
Vel Dist Location=U102-00-00      ,U102-00-00_0197 ,33548.85, 10 , 1 , 10
Vel Dist Location=U102-00-00      ,U102-00-00_0197 ,33198.41, 10 , 1 , 10
Vel Dist Location=U102-00-00      ,U102-00-00_0197 ,32860.97, 10 , 1 , 10
Vel Dist Location=U102-00-00      ,U102-00-00_0197 ,32501.36, 10 , 1 , 10
Vel Dist Location=U102-00-00      ,U102-00-00_0197 ,31927.16, 10 , 1 , 10
Vel Dist Location=U102-00-00      ,U102-00-00_0197 ,31627.03, 10 , 1 , 10
Vel Dist Location=U102-00-00      ,U102-00-00_0197 ,31554.38, 10 , 1 , 10
Vel Dist Location=U102-00-00      ,U102-00-00_0197 ,31502.26, 10 , 1 , 10
Vel Dist Location=U102-00-00      ,U102-00-00_0197 ,30893.76, 10 , 1 , 10
Vel Dist Location=U102-00-00      ,U102-00-00_0197 ,30519.31, 10 , 1 , 10
Vel Dist Location=U102-00-00      ,U102-00-00_0197 ,30460.96, 10 , 1 , 10
Vel Dist Location=U102-00-00      ,U102-00-00_0197 ,30404.01, 10 , 1 , 10
Vel Dist Location=U102-00-00      ,U102-00-00_0197 ,29758.59, 10 , 1 , 10
Vel Dist Location=U102-00-00      ,U102-00-00_0197 ,28717.43, 10 , 1 , 10
Vel Dist Location=U102-00-00      ,U102-00-00_0197 ,27577.4 , 10 , 1 , 10
Vel Dist Location=U102-00-00      ,U102-00-00_0197 ,26703.26, 10 , 1 , 10
Vel Dist Location=U102-00-00      ,U102-00-00_0197 ,25612.09, 10 , 1 , 10
Vel Dist Location=U102-00-00      ,U102-00-00_0197 ,24471.49, 10 , 1 , 10
Vel Dist Location=U102-00-00      ,U102-00-00_0197 ,24458.73, 10 , 1 , 10
Vel Dist Location=U102-00-00      ,U102-00-00_0197 ,24381.77, 10 , 1 , 10
Vel Dist Location=U102-00-00      ,U102-00-00_0197 ,24132.54, 10 , 1 , 10
Vel Dist Location=U102-00-00      ,U102-00-00_0197 ,24113.3 , 10 , 1 , 10
Vel Dist Location=U102-00-00      ,U102-00-00_0197 ,23852.4 , 10 , 1 , 10
Vel Dist Location=U102-00-00      ,U102-00-00_0197 ,23538.14, 10 , 1 , 10
Vel Dist Location=U102-00-00      ,U102-00-00_0197 ,23202.72, 10 , 1 , 10
Vel Dist Location=U102-00-00      ,U102-00-00_0197 ,22713.43, 10 , 1 , 10
Vel Dist Location=U102-00-00      ,U102-00-00_0197 ,21190.79, 10 , 1 , 10
Vel Dist Location=U102-00-00      ,U102-00-00_0197 ,20750.87, 10 , 1 , 10
Vel Dist Location=U102-00-00      ,U102-00-00_0197 ,19692.43, 10 , 1 , 10
Vel Dist Location=U102-00-00      ,U102-00-00_0197 ,20750.87, 10 , 1 , 10
Vel Dist Location=U102-00-00      ,U102-00-00_0197 ,21190.79, 10 , 1 , 10
Vel Dist Location=U102-00-00      ,U102-00-00_0197 ,22713.43, 10 , 1 , 10
Vel Dist Location=U102-00-00      ,U102-00-00_0197 ,23202.72, 10 , 1 , 10
Vel Dist Location=U102-00-00      ,U102-00-00_0197 ,23538.14, 10 , 1 , 10
Vel Dist Location=U102-00-00      ,U102-00-00_0197 ,23852.4 , 10 , 1 , 10
Vel Dist Location=U102-00-00      ,U102-00-00_0197 ,24113.3 , 10 , 1 , 10
Vel Dist Location=U102-00-00      ,U102-00-00_0197 ,24132.54, 10 , 1 , 10
Vel Dist Location=U102-00-00      ,U102-00-00_0197 ,24381.77, 10 , 1 , 10
Vel Dist Location=U102-00-00      ,U102-00-00_0197 ,24458.73, 10 , 1 , 10
Vel Dist Location=U102-00-00      ,U102-00-00_0197 ,24471.49, 10 , 1 , 10
Vel Dist Location=U102-00-00      ,U102-00-00_0197 ,25612.09, 10 , 1 , 10
Vel Dist Location=U102-00-00      ,U102-00-00_0197 ,26703.26, 10 , 1 , 10
Vel Dist Location=U102-00-00      ,U102-00-00_0197 ,27577.4 , 10 , 1 , 10
Vel Dist Location=U102-00-00      ,U102-00-00_0197 ,28717.43, 10 , 1 , 10
Vel Dist Location=U102-00-00      ,U102-00-00_0197 ,29758.59, 10 , 1 , 10
Vel Dist Location=U102-00-00      ,U102-00-00_0197 ,30404.01, 10 , 1 , 10
Vel Dist Location=U102-00-00      ,U102-00-00_0197 ,30460.96, 10 , 1 , 10
Vel Dist Location=U102-00-00      ,U102-00-00_0197 ,30519.31, 10 , 1 , 10
Vel Dist Location=U102-00-00      ,U102-00-00_0197 ,30893.76, 10 , 1 , 10
Vel Dist Location=U102-00-00      ,U102-00-00_0197 ,31502.26, 10 , 1 , 10
Vel Dist Location=U102-00-00      ,U102-00-00_0197 ,31554.38, 10 , 1 , 10
Vel Dist Location=U102-00-00      ,U102-00-00_0197 ,31627.03, 10 , 1 , 10
Vel Dist Location=U102-00-00      ,U102-00-00_0197 ,31927.16, 10 , 1 , 10
Vel Dist Location=U102-00-00      ,U102-00-00_0197 ,32501.36, 10 , 1 , 10
Vel Dist Location=U102-00-00      ,U102-00-00_0197 ,32860.97, 10 , 1 , 10
Vel Dist Location=U102-00-00      ,U102-00-00_0197 ,33198.41, 10 , 1 , 10
Vel Dist Location=U102-00-00      ,U102-00-00_0197 ,33548.85, 10 , 1 , 10
Vel Dist Location=U102-00-00      ,U102-00-00_0197 ,34772.93, 10 , 1 , 10
Vel Dist Location=U102-00-00      ,U102-00-00_0197 ,35899.56, 10 , 1 , 10
Vel Dist Location=U102-00-00      ,U102-00-00_0197 ,36534.81, 10 , 1 , 10
Vel Dist Location=U102-00-00      ,U102-00-00_0197 ,37157.18, 10 , 1 , 10
Vel Dist Location=U102-00-00      ,U102-00-00_0197 ,37207.97, 10 , 1 , 10
Vel Dist Location=U102-00-00      ,U102-00-00_0197 ,37245.13, 10 , 1 , 10
Vel Dist Location=U102-00-00      ,U102-00-00_0197 ,37416.59, 10 , 1 , 10
Vel Dist Location=U102-00-00      ,U102-00-00_0197 ,38178.64, 10 , 1 , 10
Vel Dist Location=U102-00-00      ,U102-00-00_0197 ,39300.46, 10 , 1 , 10
Vel Dist Location=U102-00-00      ,U102-00-00_0197 ,40319   , 10 , 1 , 10
Vel Dist Location=U102-00-00      ,U102-00-00_0197 ,40963.29, 10 , 1 , 10
Vel Dist Location=U102-00-00      ,U102-00-00_0197 ,41354.38, 10 , 1 , 10
Vel Dist Location=U102-00-00      ,U102-00-00_0197 ,41408.37, 10 , 1 , 10
Vel Dist Location=U102-00-00      ,U102-00-00_0197 ,41483.83, 10 , 1 , 10
Vel Dist Location=U102-00-00      ,U102-00-00_0197 ,41585.04, 10 , 1 , 10
Vel Dist Location=U102-00-00      ,U102-00-00_0197 ,42393.07, 10 , 1 , 10
Vel Dist Location=U102-00-00      ,U102-00-00_0197 ,43344.77, 10 , 1 , 10
Vel Dist Location=U102-00-00      ,U102-00-00_0197 ,44394.45, 10 , 1 , 10
Vel Dist Location=U102-00-00      ,U102-00-00_0197 ,45379.92, 10 , 1 , 10
Vel Dist Location=U102-00-00      ,U102-00-00_0197 ,45910.1 , 10 , 1 , 10
Vel Dist Location=U102-00-00      ,U102-00-00_0197 ,46304.02, 10 , 1 , 10
Vel Dist Location=U102-00-00      ,U102-00-00_0197 ,46369.31, 10 , 1 , 10
Vel Dist Location=U102-00-00      ,U102-00-00_0197 ,46387.11, 10 , 1 , 10
Vel Dist Location=U102-00-00      ,U102-00-00_0197 ,46401.06, 10 , 1 , 10
Vel Dist Location=U102-00-00      ,U102-00-00_0197 ,46507.83, 10 , 1 , 10
Vel Dist Location=U102-00-00      ,U102-00-00_0197 ,46873.4 , 10 , 1 , 10
Vel Dist Location=U102-00-00      ,U102-00-00_0197 ,46926.72, 10 , 1 , 10
Vel Dist Location=U102-00-00      ,U102-00-00_0197 ,46984.47, 10 , 1 , 10
Vel Dist Location=U102-00-00      ,U102-00-00_0197 ,47111.71, 10 , 1 , 10
Vel Dist Location=U102-00-00      ,U102-00-00_0197 ,47847.21, 10 , 1 , 10
Vel Dist Location=U102-00-00      ,U102-00-00_0197 ,48859.02, 10 , 1 , 10
Vel Dist Location=U102-00-00      ,U102-00-00_0197 ,49965.56, 10 , 1 , 10
Vel Dist Location=U102-00-00      ,U102-00-00_0197 ,50998.88, 10 , 1 , 10
Vel Dist Location=U102-00-00      ,U102-00-00_0197 ,51047.25, 10 , 1 , 10
Vel Dist Location=U102-00-00      ,U102-00-00_0197 ,51146.17, 10 , 1 , 10
Vel Dist Location=U102-00-00      ,U102-00-00_0197 ,51782.55, 10 , 1 , 10
Vel Dist Location=U102-00-00      ,U102-00-00_0197 ,51929.68, 10 , 1 , 10
Vel Dist Location=U102-00-00      ,U102-00-00_0197 ,52014.66, 10 , 1 , 10
Vel Dist Location=U102-00-00      ,U102-00-00_0197 ,52072.36, 10 , 1 , 10
Vel Dist Location=U102-00-00      ,U102-00-00_0197 ,52104.96, 10 , 1 , 10
Vel Dist Location=U102-00-00      ,U102-00-00_0197 ,52204.51, 10 , 1 , 10
Vel Dist Location=U102-00-00      ,U102-00-00_0197 ,52414.93, 10 , 1 , 10
Vel Dist Location=U102-00-00      ,U102-00-00_0197 ,53109.38, 10 , 1 , 10
Vel Dist Location=U102-00-00      ,U102-00-00_0197 ,54244.41, 10 , 1 , 10
Vel Dist Location=U102-00-00      ,U102-00-00_0197 ,54885.61, 10 , 1 , 10
Vel Dist Location=U102-00-00      ,U102-00-00_0197 ,55351.98, 10 , 1 , 10
Vel Dist Location=U102-00-00      ,U102-00-00_0197 ,55580.36, 10 , 1 , 10
Vel Dist Location=U102-00-00      ,U102-00-00_0197 ,55887.13, 10 , 1 , 10
Vel Dist Location=U102-00-00      ,U102-00-00_0197 ,56132.66, 10 , 1 , 10
Vel Dist Location=U102-00-00      ,U102-00-00_0197 ,56194.89, 10 , 1 , 10
Vel Dist Location=U102-00-00      ,U102-00-00_0197 ,56470.21, 10 , 1 , 10
Vel Dist Location=U102-00-00      ,U102-00-00_0197 ,56666.18, 10 , 1 , 10
Vel Dist Location=U102-00-00      ,U102-00-00_0197 ,56832.31, 10 , 1 , 10
Vel Dist Location=U102-00-00      ,U102-00-00_0197 ,57037.9 , 10 , 1 , 10
Vel Dist Location=U102-00-00      ,U102-00-00_0197 ,57093.08, 10 , 1 , 10
Vel Dist Location=U102-00-00      ,U102-00-00_0197 ,57213.66, 10 , 1 , 10
Vel Dist Location=U102-00-00      ,U102-00-00_0197 ,58086.16, 10 , 1 , 10
Vel Dist Location=U102-00-00      ,U102-00-00_0197 ,59168.92, 10 , 1 , 10
Vel Dist Location=U102-00-00      ,U102-00-00_0197 ,60176.11, 10 , 1 , 10
Vel Dist Location=U102-00-00      ,U102-00-00_0197 ,61507.56, 10 , 1 , 10
Vel Dist Location=U102-00-00      ,U102-00-00_0197 ,62613.3 , 10 , 1 , 10
Vel Dist Location=U102-00-00      ,U102-00-00_0197 ,63182.11, 10 , 1 , 10
Vel Dist Location=U102-00-00      ,U102-00-00_0197 ,63435.61, 10 , 1 , 10
Vel Dist Location=U102-00-00      ,U102-00-00_0197 ,63482.86, 10 , 1 , 10
Vel Dist Location=U102-00-00      ,U102-00-00_0197 ,63543.31, 10 , 1 , 10
Vel Dist Location=U102-00-00      ,U102-00-00_0197 ,63598.3 , 10 , 1 , 10
Vel Dist Location=U102-00-00      ,U102-00-00_0197 ,64170.07, 10 , 1 , 10
Vel Dist Location=U102-00-00      ,U102-00-00_0197 ,65139.42, 10 , 1 , 10
Vel Dist Location=U102-00-00      ,U102-00-00_0197 ,65864.54, 10 , 1 , 10
Vel Dist Location=U102-00-00      ,U102-00-00_0197 ,66253.16, 10 , 1 , 10
Vel Dist Location=U102-00-00      ,U102-00-00_0197 ,67625.08, 10 , 1 , 10
Vel Dist Location=U102-00-00      ,U102-00-00_0197 ,68441.07, 10 , 1 , 10
Vel Dist Location=U102-00-00      ,U102-00-00_0197 ,68877.77, 10 , 1 , 10
Vel Dist Location=U102-00-00      ,U102-00-00_0197 ,68899.68, 10 , 1 , 10
Vel Dist Location=U102-00-00      ,U102-00-00_0197 ,68924.32, 10 , 1 , 10
Vel Dist Location=U102-00-00      ,U102-00-00_0197 ,69031.07, 10 , 1 , 10
Vel Dist Location=U102-00-00      ,U102-00-00_0197 ,69870.13, 10 , 1 , 10
Vel Dist Location=U102-00-00      ,U102-00-00_0197 ,71324.16, 10 , 1 , 10
Vel Dist Location=U102-00-00      ,U102-00-00_0197 ,71949.68, 10 , 1 , 10
Vel Dist Location=U102-00-00      ,U102-00-00_0197 ,73108.58, 10 , 1 , 10
Vel Dist Location=U102-00-00      ,U102-00-00_0197 ,74313.45, 10 , 1 , 10
Vel Dist Location=U102-00-00      ,U102-00-00_0197 ,74758.11, 10 , 1 , 10
Vel Dist Location=U102-00-00      ,U102-00-00_0197 ,76413.3 , 10 , 1 , 10
Vel Dist Location=U102-00-00      ,U102-00-00_0197 ,77603.52, 10 , 1 , 10
Vel Dist Location=U102-00-00      ,U102-00-00_0197 ,78422.85, 10 , 1 , 10
Vel Dist Location=U102-00-00      ,U102-00-00_0197 ,78654.82, 10 , 1 , 10
Vel Dist Location=U102-00-00      ,U102-00-00_0197 ,78672.98, 10 , 1 , 10
Vel Dist Location=U102-00-00      ,U102-00-00_0197 ,78687.62, 10 , 1 , 10
Vel Dist Location=U102-00-00      ,U102-00-00_0197 ,78904.98, 10 , 1 , 10
Vel Dist Location=U102-00-00      ,U102-00-00_0197 ,80119.4 , 10 , 1 , 10
Vel Dist Location=U102-00-00      ,U102-00-00_0197 ,81073.43, 10 , 1 , 10
Vel Dist Location=U102-00-00      ,U102-00-00_0197 ,81731.22, 10 , 1 , 10
Vel Dist Location=U102-00-00      ,U102-00-00_0197 ,82591.49, 10 , 1 , 10
Global Log Level= 0
CheckData=True
Encroach Param=-1 ,0,0, 2
Encroach River=U102-00-00
Encroach Reach=U102-00-00_0197
Encroach Node=82591.49
       1 3797.94 9294.98
Encroach Node=81731.22
       1 3743.44 8789.76
Encroach Node=81073.43
       1 4146.85 8218.86
Encroach Node=80119.4
       1 5297.11 8081.26
Encroach Node=78904.98
       1 5767.11 7670.39
Encroach Node=78687.62
       1  6799.4 8433.22
Encroach Node=78654.82
       1    6666 8462.04
Encroach Node=78422.85
       1 6836.01 8568.32
Encroach Node=77603.52
       1 7600.85 9147.44
Encroach Node=76413.3
       1 6769.15 8339.68
Encroach Node=74758.11
       1 6472.97 8699.84
Encroach Node=74313.45
       1 7389.25 9280.23
Encroach Node=73108.58
       1 8012.5910470.83
Encroach Node=71949.68
       1 9148.97 11214.4
Encroach Node=71324.16
       1 9888.2911701.93
Encroach Node=69870.13
       1  9113.810636.73
Encroach Node=69031.07
       1 8226.07 9314.17
Encroach Node=68924.32
       1 7095.46    9196
Encroach Node=68877.77
       1    7010  9135.8
Encroach Node=68441.07
       1    6516 8546.17
Encroach Node=67625.08
       1 6198.77  8491.9
Encroach Node=66253.16
       1 6385.56 8418.97
Encroach Node=65864.54
       1 6322.07 8254.99
Encroach Node=65139.42
       1 6161.87 8289.26
Encroach Node=64170.07
       1    6658 8350.06
Encroach Node=63598.3
       1 6868.63 8373.14
Encroach Node=63543.31
       1    6868    8585
Encroach Node=63435.61
       1 6850.12 8584.14
Encroach Node=63182.11
       1 6902.27 8615.27
Encroach Node=62613.3
       1 7061.44 8684.28
Encroach Node=61507.56
       1 7090.43 9176.47
Encroach Node=60176.11
       1 7086.82 9408.62
Encroach Node=59168.92
       1 3864.16 5432.35
Encroach Node=58086.16
       1 3872.03    5329
Encroach Node=57213.66
       1 4233.76    5355
Encroach Node=57093.08
       1 3959.33 5291.12
Encroach Node=57037.9
       1 3912.72    5255
Encroach Node=56832.31
       1 3884.72 5300.58
Encroach Node=56666.18
       1 4060.52 5294.44
Encroach Node=56470.21
       1 4110.67 5275.07
Encroach Node=56194.89
       1 4100.06 5274.84
Encroach Node=56132.66
       1 4084.76 5250.26
Encroach Node=55887.13
       1 4361.06 5161.69
Encroach Node=55580.36
       1 4444.97 5069.92
Encroach Node=55351.98
       1 4606.58 5131.03
Encroach Node=54885.61
       1 2698.11 2924.17
Encroach Node=54244.41
       1 2169.34 2321.92
Encroach Node=53109.38
       1 4446.19 4592.53
Encroach Node=52414.93
       1 4277.47 4431.54
Encroach Node=52204.51
       1 4269.68 4433.68
Encroach Node=52104.96
       1 4342.53 4548.89
Encroach Node=52014.66
       1 4362.17 4539.06
Encroach Node=51929.68
       1 4281.09 4497.69
Encroach Node=51782.55
       1 4321.44 4520.92
Encroach Node=51146.17
       1  3903.5 4129.87
Encroach Node=50998.88
       1 3963.46 4139.79
Encroach Node=49965.56
       1 3452.23 3599.82
Encroach Node=48859.02
       1 2501.05 2629.06
Encroach Node=47847.21
       1 2057.92 2239.85
Encroach Node=47111.71
       1 1861.37 2014.37
Encroach Node=46984.47
       1 1645.46 1779.37
Encroach Node=46873.4
       1 1645.46 1774.42
Encroach Node=46507.83
       1 2022.65 2186.74
Encroach Node=46401.06
       1  1988.9  2156.9
Encroach Node=46387.11
       1 2074.44  2240.4
Encroach Node=46369.31
       1 2074.44  2240.4
Encroach Node=46304.02
       1 2064.55 2230.64
Encroach Node=45910.1
       1 1994.46 2193.63
Encroach Node=45379.92
       1 1767.77 1923.81
Encroach Node=44394.45
       1 1824.25 1972.72
Encroach Node=43344.77
       1 1732.72 1883.76
Encroach Node=42393.07
       1 1411.83 1578.72
Encroach Node=41585.04
       1 1862.17 2009.96
Encroach Node=41483.83
       1 1771.96 1934.77
Encroach Node=41354.38
       1 1786.86 1944.53
Encroach Node=40963.29
       1 1219.99 1388.92
Encroach Node=40319
       1 2665.81 2835.93
Encroach Node=39300.46
       1  2806.8 2983.28
Encroach Node=38178.64
       1 2438.81 2608.03
Encroach Node=37416.59
       1 1044.05 1207.82
Encroach Node=37245.13
       1 1253.17 1405.84
Encroach Node=37157.18
       1 1233.62 1405.84
Encroach Node=36534.81
       1 1971.09 2140.77
Encroach Node=35899.56
       1 1857.35 2032.23
Encroach Node=34772.93
       1 2081.87 2319.51
Encroach Node=33548.85
       1 2194.66 2455.06
Encroach Node=33198.41
       1  1586.1 2314.43
Encroach Node=32860.97
       1 1584.42 2103.68
Encroach Node=32501.36
       1 1727.93 1890.68
Encroach Node=31927.16
       1  949.51 1118.31
Encroach Node=31627.03
       1  779.07  973.43
Encroach Node=31502.26
       1  798.98 1038.33
Encroach Node=30893.76
       1 1155.21 1374.12
Encroach Node=30519.31
       1 1128.69 1342.58
Encroach Node=30404.01
       1 1158.66  1357.4
Encroach Node=29758.59
       1 1303.23 1487.27
Encroach Node=28717.43
       1 2435.92 2632.93
Encroach Node=27577.4
       1 2857.58 3028.98
Encroach Node=25612.09
       1 2836.66 2959.83
Encroach Node=24471.49
       1 3413.83 3603.61
Encroach Node=24458.73
       1 3433.81 3623.59
Encroach Node=24381.77
       1 3413.79 3593.61
Encroach Node=24132.54
       1 3527.39 3707.18
Encroach Node=24113.3
       1 3562.35 3747.12
Encroach Node=23852.4
       1 3421.54 3616.26
Encroach Node=23538.14
       1 3163.75  3358.4
Encroach Node=23202.72
       1 2894.84 3089.83
Encroach Node=22713.43
       1 3421.05 3625.58
Encroach Node=21190.79
       1 1488.01 3219.76
Encroach Node=20750.87
       1 1492.21 3217.74
Encroach Node=19692.43
       1 1588.33 3107.28
BEGIN DESCRIPTION:
FEMA Effective Floodway November 2019 + LOMR 20-06-2070P
Post-Project Condition
END DESCRIPTION:
Computation Interval=1HOUR
Output Interval=1HOUR
Run HTab= 0
Run UNet= 0
Run PostProcess= 0
Run WQNet= 0
UNET Theta= 1
UNET Theta Warmup= 1
UNET ZTol= 0.02
UNET ZSATol= 0.05
UNET MxIter= 20
UNET MaxInSteps= 0
UNET DtIC= 0
UNET DtMin= 0
UNET MaxCRTS= 20
UNET WFStab= 2
UNET SFStab= 1
UNET WFX= 1
UNET SFX= 1
UNET DSS MLevel= 4
UNET DZMax Abort= 100
UNET Convert EG Bridges= 0
UNET Use Existing IB Tables=-1
UNET Froude Reduction=False
UNET Froude Limit= 1
UNET Froude Power= 10
UNET Time Slicing=0,0, 5
UNET Junction Losses=0
Instantaneous Interval=1HOUR
Write IC File= 0
Write IC File at Sim End=0
Echo Input=False
Echo Parameters=False
Echo Output=False
Write Detailed= 0
WQ AD Non Conservative
WQ ULTIMATE=-1
WQ Max Comp Step=1HOUR
WQ Output Interval=15MIN
WQ Output Selected Increments= 0
WQ Output face flow=0
WQ Output face velocity=0
WQ Output face area=0
WQ Output face dispersion=0
WQ Output cell volume=0
WQ Output cell surface area=0
WQ Output cell continuity=0
WQ Output cumulative cell continuity=0
WQ Output face conc=0
WQ Output face dconc_dx=0
WQ Output face courant=0
WQ Output face peclet=0
WQ Output face adv mass=0
WQ Output face disp mass=0
WQ Output cell mass=0
WQ Output cell source sink temp=0
WQ Output cell source sink nsm=0
WQ Output MaxMinRange=-1
WQ Daily Max Min Mean=-1
WQ Daily Range=0
WQ Daily Time=0
WQ Create Restart=0
WQ Fixed Restart=0
WQ System Summary=0
WQ Use Fixed Temperature=0
Sorting and Armoring Iterations= 10
XS Update Threshold= 0.02
Hydraulics Update Threshold= 0.02
Energy Slope Method= 1
Volume Change Method= 0
XS Weighting Method= 0
Number of US Weighted Cross Sections= 1
Number of DS Weighted Cross Sections= 1
Upstream XS Weight=0.25
Main XS Weight=0.5
Downstream XS Weight=0.25
Number of DS XS's Weighted with US Boundary= 1
Upstream Boundary Weight= 1
Weight of XSs Associated with US Boundary= 0
Number of US XS's Weighted with DS Boundary= 1
Downstream Boundary Weight= 0.5
Weight of XSs Associated with DS Boundary= 0.5
Sediment Output Level= 4
Mass or Volume Output= 0
Output Increment Type= 1
Profile and TS Output Increment= 10
XS Output Flag= 0
XS Output Increment= 10
Disregard all LS=0
Disregard all Conn=0
Disregard all Breaches=0
Disregard all Pumps=0

--- U102-00-00.f01 (steady flow) ---

Flow Title=Effective Multi-Profile 2020 (Re-Study)
Program Version=4.10
Number of Profiles= 4
Profile Names=10YR,50YR,100YR,500YR
River Rch & RM=U102-00-00,U102-00-00_0197 ,82591.49
    1723    4535    6535   13230
River Rch & RM=U102-00-00,U102-00-00_0197 ,81073.43
    1708    4419    6347   12634
River Rch & RM=U102-00-00,U102-00-00_0197 ,80119.4
    1688    4274    6115   11914
River Rch & RM=U102-00-00,U102-00-00_0197 ,78904.98
    1667    4125    5877   11188
River Rch & RM=U102-00-00,U102-00-00_0197 ,77603.52
    1648    3992    5667   10563
River Rch & RM=U102-00-00,U102-00-00_0197 ,76413.3
    1622    3816    5387    9751
River Rch & RM=U102-00-00,U102-00-00_0197 ,74758.11
    1615    3769    5314    9544
River Rch & RM=U102-00-00,U102-00-00_0197 ,74313.45
    1596    3647    5122    9004
River Rch & RM=U102-00-00,U102-00-00_0197 ,73108.58
    1578    3533    4944    8514
River Rch & RM=U102-00-00,U102-00-00_0197 ,71949.68
    1569    3473    4850    8260
River Rch & RM=U102-00-00,U102-00-00_0197 ,71324.16
    1547    3338    4639    7700
River Rch & RM=U102-00-00,U102-00-00_0197 ,69870.13
    1526    3210    4440    7186
River Rch & RM=U102-00-00,U102-00-00_0197 ,68441.07
    1514    3139    4331    6909
River Rch & RM=U102-00-00,U102-00-00_0197 ,67625.08
    1494    3023    4153    6466
River Rch & RM=U102-00-00,U102-00-00_0197 ,66253.16
    1478    2933    4014    6127
River Rch & RM=U102-00-00,U102-00-00_0197 ,65139.42
    1456    2807    3823    5672
River Rch & RM=U102-00-00,U102-00-00_0197 ,63543.31
    1451    2780    3781    5574
River Rch & RM=U102-00-00,U102-00-00_0197 ,63182.11
    1513    2875    3864    5678
River Rch & RM=U102-00-00,U102-00-00_0197 ,61507.56
    1564    2952    3931    5762
River Rch & RM=U102-00-00,U102-00-00_0197 ,60176.11
    1604    3012    3983    5826
River Rch & RM=U102-00-00,U102-00-00_0197 ,59168.92
    1648    3079    4039    5896
River Rch & RM=U102-00-00,U102-00-00_0197 ,58086.16
    1716    3180    4125    6001
River Rch & RM=U102-00-00,U102-00-00_0197 ,56470.21
    1785    3282    4210    6107
River Rch & RM=U102-00-00,U102-00-00_0197 ,54885.61
    1814    3325    4245    6150
River Rch & RM=U102-00-00,U102-00-00_0197 ,54244.41
    1866    3401    4308    6227
River Rch & RM=U102-00-00,U102-00-00_0197 ,53109.38
    1929    3493    4383    6319
River Rch & RM=U102-00-00,U102-00-00_0197 ,51782.55
    1960    3538    4419    6363
River Rch & RM=U102-00-00,U102-00-00_0197 ,51146.17
    2019    3623    4488    6447
River Rch & RM=U102-00-00,U102-00-00_0197 ,49965.56
    2076    3704    4553    6525
River Rch & RM=U102-00-00,U102-00-00_0197 ,48859.02
    2129    3780    4613    6599
River Rch & RM=U102-00-00,U102-00-00_0197 ,47847.21
    2202    3882    4694    6697
River Rch & RM=U102-00-00,U102-00-00_0197 ,46507.83
    2309    4083    4939    7086
River Rch & RM=U102-00-00,U102-00-00_0197 ,43344.77
    2416    4285    5187    7479
River Rch & RM=U102-00-00,U102-00-00_0197 ,40319
    2530    4500    5450    7901
River Rch & RM=U102-00-00,U102-00-00_0197 ,37245.13
    2626    4681    5672    8257
River Rch & RM=U102-00-00,U102-00-00_0197 ,34772.93
    2753    4922    5968    8734
River Rch & RM=U102-00-00,U102-00-00_0197 ,31627.03
    2876    5155    6255    9200
River Rch & RM=U102-00-00,U102-00-00_0197 ,28717.43
    3014    5417    6576    9724
River Rch & RM=U102-00-00,U102-00-00_0197 ,25612.09
    3125    5629    6837   10152
River Rch & RM=U102-00-00,U102-00-00_0197 ,23202.72
    3677    6531    7993   12116
River Rch & RM=U102-00-00,U102-00-00_0197 ,22713.43
    3654    6385    7802   11956
River Rch & RM=U102-00-00,U102-00-00_0197 ,21190.79
    3632    6244    7618   11801
Boundary for River Rch & Prof#=U102-00-00,U102-00-00_0197 , 1
Up Type= 0
Dn Type= 1
Dn Known WS=97.6
Boundary for River Rch & Prof#=U102-00-00,U102-00-00_0197 , 2
Up Type= 0
Dn Type= 1
Dn Known WS=99.9
Boundary for River Rch & Prof#=U102-00-00,U102-00-00_0197 , 3
Up Type= 0
Dn Type= 1
Dn Known WS=100.8
Boundary for River Rch & Prof#=U102-00-00,U102-00-00_0197 , 4
Up Type= 0
Dn Type= 1
Dn Known WS=102.4
Observed WS=U102-00-00      ,U102-00-00_0197 ,82591.49,0,158.16,159.06,159.67,160.72
Observed WS=U102-00-00      ,U102-00-00_0197 ,81731.22,0,158.01,158.96,159.56,160.61
Observed WS=U102-00-00      ,U102-00-00_0197 ,81073.43,0,157.89,158.87,159.46,160.5
Observed WS=U102-00-00      ,U102-00-00_0197 ,80119.4 ,0,157.43,158.58,159.15,160.22
Observed WS=U102-00-00      ,U102-00-00_0197 ,78904.98,0,156.64,157.98,158.54,159.41
Observed WS=U102-00-00      ,U102-00-00_0197 ,78687.62,0,156.43,157.74,158.18,159.22
Observed WS=U102-00-00      ,U102-00-00_0197 ,78654.82,0,156.28,157.62,158.22,159.07
Observed WS=U102-00-00      ,U102-00-00_0197 ,78422.85,0,156.08,157.26,158.07,158.84
Observed WS=U102-00-00      ,U102-00-00_0197 ,77603.52,0,155.6,156.75,157.6,158.07
Observed WS=U102-00-00      ,U102-00-00_0197 ,76413.3 ,0,154.81,155.74,156.5,157
Observed WS=U102-00-00      ,U102-00-00_0197 ,74758.11,0,153.89,154.79,154.95,156.08
Observed WS=U102-00-00      ,U102-00-00_0197 ,74313.45,0,153.53,154.42,154.69,155.7
Observed WS=U102-00-00      ,U102-00-00_0197 ,73108.58,0,152.52,153.47,153.8,155.25
Observed WS=U102-00-00      ,U102-00-00_0197 ,71949.68,0,151.23,152.18,152.72,153.59
Observed WS=U102-00-00      ,U102-00-00_0197 ,71324.16,0,150.35,151.52,152.24,153.02
Observed WS=U102-00-00      ,U102-00-00_0197 ,69870.13,0,149.28,150.04,150.44,152.19
Observed WS=U102-00-00      ,U102-00-00_0197 ,69031.07,0,148.94,149.64,149.91,151.5
Observed WS=U102-00-00      ,U102-00-00_0197 ,68924.32,0,148.84,149.46,149.61,151.34
Observed WS=U102-00-00      ,U102-00-00_0197 ,68877.77,0,148.38,149.14,149.53,151.13
Observed WS=U102-00-00      ,U102-00-00_0197 ,68441.07,0,148.05,148.79,149.14,150.67
Observed WS=U102-00-00      ,U102-00-00_0197 ,67625.08,0,147.5,148.29,148.61,150
Observed WS=U102-00-00      ,U102-00-00_0197 ,66253.16,0,146.34,147.21,147.51,148.64
Observed WS=U102-00-00      ,U102-00-00_0197 ,65864.54,0,146.04,146.77,147.03,148.22
Observed WS=U102-00-00      ,U102-00-00_0197 ,65139.42,0,145.46,146.17,146.43,147.74
Observed WS=U102-00-00      ,U102-00-00_0197 ,64170.07,0,144.7,145.61,145.82,147.13
Observed WS=U102-00-00      ,U102-00-00_0197 ,63598.3 ,0,144.41,145.37,145.53,146.69
Observed WS=U102-00-00      ,U102-00-00_0197 ,63543.31,0,144.42,145.37,145.53,146.67
Observed WS=U102-00-00      ,U102-00-00_0197 ,63435.61,0,144.37,144.97,145.22,146.6
Observed WS=U102-00-00      ,U102-00-00_0197 ,63182.11,0,144.2,144.81,145.07,146.47
Observed WS=U102-00-00      ,U102-00-00_0197 ,62613.3 ,0,143.73,144.41,144.68,146.11
Observed WS=U102-00-00      ,U102-00-00_0197 ,61507.56,0,143.15,143.84,144.11,145.45
Observed WS=U102-00-00      ,U102-00-00_0197 ,60176.11,0,142.48,143.23,143.54,144.71
Observed WS=U102-00-00      ,U102-00-00_0197 ,59168.92,0,141.94,142.74,143.07,144.16
Observed WS=U102-00-00      ,U102-00-00_0197 ,58086.16,0,141.36,142.12,142.42,143.66
Observed WS=U102-00-00      ,U102-00-00_0197 ,57213.66,0,140.83,141.31,141.46,143.16
Observed WS=U102-00-00      ,U102-00-00_0197 ,57093.08,0,140.71,140.99,140.95,142.08
Observed WS=U102-00-00      ,U102-00-00_0197 ,57037.9 ,0,136.95,139.28,139.97,141.95
Observed WS=U102-00-00      ,U102-00-00_0197 ,56832.31,0,136.92,139.23,139.89,141.85
Observed WS=U102-00-00      ,U102-00-00_0197 ,56666.18,0,136.69,139.02,139.66,141.74
Observed WS=U102-00-00      ,U102-00-00_0197 ,56470.21,0,136.41,138.77,139.39,141.6
Observed WS=U102-00-00      ,U102-00-00_0197 ,56194.89,0,135.49,137.8,138.2,141.47
Observed WS=U102-00-00      ,U102-00-00_0197 ,56132.66,0,135.2,137.52,138.32,141.35
Observed WS=U102-00-00      ,U102-00-00_0197 ,55887.13,0,134.52,136.85,137.71,140.96
Observed WS=U102-00-00      ,U102-00-00_0197 ,55580.36,0,133.67,136.01,136.94,140.47
Observed WS=U102-00-00      ,U102-00-00_0197 ,55351.98,0,133.04,135.39,136.37,140.11
Observed WS=U102-00-00      ,U102-00-00_0197 ,54885.61,0,132.59,134.99,136,139.62
Observed WS=U102-00-00      ,U102-00-00_0197 ,54244.41,0,131.97,134.45,135.48,138.94
Observed WS=U102-00-00      ,U102-00-00_0197 ,53109.38,0,130.86,133.41,134.44,137.96
Observed WS=U102-00-00      ,U102-00-00_0197 ,52414.93,0,130.45,133.04,134.07,137.55
Observed WS=U102-00-00      ,U102-00-00_0197 ,52204.51,0,130.33,132.92,133.96,137.43
Observed WS=U102-00-00      ,U102-00-00_0197 ,52104.96,0,130.27,132.87,133.91,137.37
Observed WS=U102-00-00      ,U102-00-00_0197 ,52014.66,0,130.22,132.82,133.86,137.3
Observed WS=U102-00-00      ,U102-00-00_0197 ,51929.68,0,130.18,132.78,133.82,137.23
Observed WS=U102-00-00      ,U102-00-00_0197 ,51782.55,0,130.11,132.7,133.74,137.12
Observed WS=U102-00-00      ,U102-00-00_0197 ,51146.17,0,129.79,132.37,133.4,136.63
Observed WS=U102-00-00      ,U102-00-00_0197 ,50998.88,0,129.67,132.25,133.27,136.54
Observed WS=U102-00-00      ,U102-00-00_0197 ,49965.56,0,128.86,131.37,132.32,135.87
Observed WS=U102-00-00      ,U102-00-00_0197 ,48859.02,0,127.64,130.07,131.04,135.17
Observed WS=U102-00-00      ,U102-00-00_0197 ,47847.21,0,126.34,128.74,129.68,134.35
Observed WS=U102-00-00      ,U102-00-00_0197 ,47111.71,0,125.62,128.08,128.98,133.79
Observed WS=U102-00-00      ,U102-00-00_0197 ,46984.47,0,124.9,127.09,127.75,131.25
Observed WS=U102-00-00      ,U102-00-00_0197 ,46873.4 ,0,124.69,126.85,127.48,129.97
Observed WS=U102-00-00      ,U102-00-00_0197 ,46507.83,0,124.75,126.99,127.66,130.74
Observed WS=U102-00-00      ,U102-00-00_0197 ,46401.06,0,124.68,126.9,127.55,130.67
Observed WS=U102-00-00      ,U102-00-00_0197 ,46387.11,0,124.69,126.91,127.57,130.46
Observed WS=U102-00-00      ,U102-00-00_0197 ,46369.31,0,122.29,124.72,125.8,130.41
Observed WS=U102-00-00      ,U102-00-00_0197 ,46304.02,0,122.28,124.71,125.8,130.41
Observed WS=U102-00-00      ,U102-00-00_0197 ,45910.1 ,0,122.21,124.67,125.77,130.42
Observed WS=U102-00-00      ,U102-00-00_0197 ,45379.92,0,121.81,124.2,125.28,129.88
Observed WS=U102-00-00      ,U102-00-00_0197 ,44394.45,0,120.84,123.15,124.18,128.82
Observed WS=U102-00-00      ,U102-00-00_0197 ,43344.77,0,119.68,121.93,122.95,127.43
Observed WS=U102-00-00      ,U102-00-00_0197 ,42393.07,0,118.22,120.51,121.55,126.11
Observed WS=U102-00-00      ,U102-00-00_0197 ,41585.04,0,117.3,119.54,120.56,124.66
Observed WS=U102-00-00      ,U102-00-00_0197 ,41483.83,0,117.2,119.44,120.46,124.49
Observed WS=U102-00-00      ,U102-00-00_0197 ,41354.38,0,116.88,119.07,120.07,124.2
Observed WS=U102-00-00      ,U102-00-00_0197 ,40963.29,0,116.62,118.81,119.82,123.93
Observed WS=U102-00-00      ,U102-00-00_0197 ,40319   ,0,116.03,118.19,119.19,123.33
Observed WS=U102-00-00      ,U102-00-00_0197 ,39300.46,0,115.16,117.35,118.37,122.45
Observed WS=U102-00-00      ,U102-00-00_0197 ,38178.64,0,114.19,116.38,117.4,121.47
Observed WS=U102-00-00      ,U102-00-00_0197 ,37416.59,0,113.67,115.77,116.77,120.45
Observed WS=U102-00-00      ,U102-00-00_0197 ,37245.13,0,113.52,115.58,116.57,120.04
Observed WS=U102-00-00      ,U102-00-00_0197 ,37157.18,0,113.36,115.4,116.37,119.85
Observed WS=U102-00-00      ,U102-00-00_0197 ,36534.81,0,112.53,114.61,115.62,118.84
Observed WS=U102-00-00      ,U102-00-00_0197 ,35899.56,0,111.76,113.95,115,117.96
Observed WS=U102-00-00      ,U102-00-00_0197 ,34772.93,0,110.1,112.59,113.75,116.39
Observed WS=U102-00-00      ,U102-00-00_0197 ,33548.85,0,109.65,112.22,113.39,115.88
Observed WS=U102-00-00      ,U102-00-00_0197 ,33198.41,0,109.44,111.99,113.15,115.41
Observed WS=U102-00-00      ,U102-00-00_0197 ,32860.97,0,109.24,111.76,112.91,114.95
Observed WS=U102-00-00      ,U102-00-00_0197 ,32501.36,0,109.03,111.52,112.66,114.47
Observed WS=U102-00-00      ,U102-00-00_0197 ,31927.16,0,108.96,111.48,112.64,114.5
Observed WS=U102-00-00      ,U102-00-00_0197 ,31627.03,0,108.89,111.4,112.56,114.35
Observed WS=U102-00-00      ,U102-00-00_0197 ,31502.26,0,108.77,111.28,112.43,114.09
Observed WS=U102-00-00      ,U102-00-00_0197 ,30893.76,0,108.59,111.08,112.23,113.71
Observed WS=U102-00-00      ,U102-00-00_0197 ,30519.31,0,108.48,110.95,112.1,113.49
Observed WS=U102-00-00      ,U102-00-00_0197 ,30404.01,0,108.32,110.88,112.01,113.38
Observed WS=U102-00-00      ,U102-00-00_0197 ,29758.59,0,107.88,110.38,111.5,112.84
Observed WS=U102-00-00      ,U102-00-00_0197 ,28717.43,0,107.33,109.8,110.9,111.63
Observed WS=U102-00-00      ,U102-00-00_0197 ,27577.4 ,0,106.66,109.05,110.12,110.74
Observed WS=U102-00-00      ,U102-00-00_0197 ,26703.26,0,105.75,107.95,108.94,109.98
Observed WS=U102-00-00      ,U102-00-00_0197 ,25612.09,0,103.3,104.73,105.35,107.96
Observed WS=U102-00-00      ,U102-00-00_0197 ,24471.49,0,102.93,104.3,104.93,106.84
Observed WS=U102-00-00      ,U102-00-00_0197 ,24458.73,0,102.92,104.29,104.91,106.81
Observed WS=U102-00-00      ,U102-00-00_0197 ,24381.77,0,102.87,104.2,104.81,106.65
Observed WS=U102-00-00      ,U102-00-00_0197 ,24132.54,0,102.7,103.94,104.49,106.14
Observed WS=U102-00-00      ,U102-00-00_0197 ,24113.3 ,0,102.69,103.92,104.47,106.1
Observed WS=U102-00-00      ,U102-00-00_0197 ,23852.4 ,0,102.6,103.78,104.31,105.76
Observed WS=U102-00-00      ,U102-00-00_0197 ,23538.14,0,102.5,103.61,104.11,105.36
Observed WS=U102-00-00      ,U102-00-00_0197 ,23202.72,0,102.37,103.43,103.91,105.21
Observed WS=U102-00-00      ,U102-00-00_0197 ,22713.43,0,102.27,103.28,103.74,104.97
Observed WS=U102-00-00      ,U102-00-00_0197 ,21190.79,0,101.8,102.66,103.07,104.2
Observed WS=U102-00-00      ,U102-00-00_0197 ,20750.87,0,101.65,102.46,102.86,103.97
Observed WS=U102-00-00      ,U102-00-00_0197 ,19692.43,0,98.2,99.9,100.8,102.4
DSS Import GetInterval= 0
DSS Import GetPeak= 0
DSS Import FillOption= 0
